HEC-RAS study PROCTRCK.prj: PROCTRCK

--- PROCTRCK.g01 (geometry) --- (continued)

Type RM Length L Ch R = 1 ,22249   ,640.7,627.7,630.9
XS GIS Cut Line= 3
1607024.88448804432640.5027531441606971.33035849 432771.41284759
1606689.67530681433088.770652309
#Sta/Elev= 30
       0  849.88    34.4  839.59   116.7  822.44   148.3  813.48   175.7   803.4
   196.4  789.05   212.6  781.07   223.2  777.62   229.5  777.11   240.9  779.05
     266   778.7   274.9   777.9   287.3   778.5   335.5  777.13   351.4  777.34
   368.4  776.18   387.5772.4542   399.5  771.22   417.5  771.38   423.5  772.39
   430.7  775.96   437.1  781.67   442.4  785.41   463.8   792.7   473.2  795.14
   513.9  811.39   533.4  824.25   549.4   836.5   554.8  840.85   565.8  851.25
#Mann= 5, -1 ,  0
       0     0.1       0  371.44    0.06       0   387.5   0.045       0
   423.5    0.06       0  521.44     0.1       0
Bank Sta=387.5,423.5
XS Rating Curve= 0 ,0
Exp/Cntr(USF)=0,0
Exp/Cntr=0.3,0.1

Type RM Length L Ch R = 1 ,21621   ,407.2,392.5,385.4
XS GIS Cut Line= 4
1606507.19456909432335.045866102 1606497.2771377432410.418344723
1606437.77254931432709.9247729261606441.73952187432878.521106683
#Sta/Elev= 30
       0  868.74    13.6  869.24    29.7  868.47    33.8  867.37      40  863.48
    53.9  850.44      62  841.33    78.2  812.78    99.2  784.99   110.8  772.49
   114.9  769.07   125.8766.0778   135.3  765.21   151.6  766.06   176.1  766.04
   192.4  771.24   204.6  771.57   212.8  772.78   237.2  770.57   249.5  771.86
   273.9  771.71   318.8  773.81   367.7  774.62     412  773.85     432  774.83
     444  776.94   496.4  791.15   530.9  808.52   537.4  813.58     550  825.15
#Mann= 5, -1 ,  0
       0     0.1       0   125.8   0.045       0   151.6     0.1       0
  166.02    0.06       0  266.02     0.1       0
Bank Sta=125.8,151.6
XS Rating Curve= 0 ,0
Exp/Cntr(USF)=0,0
Exp/Cntr=0.3,0.1

Type RM Length L Ch R = 1 ,21229   ,426.5,419.4,415.4
XS GIS Cut Line= 3
1606049.73539827432431.7895704611606219.03159039432791.543978722
  1606267.401931432903.400391374
#Sta/Elev= 30
       0  835.79     5.2  829.26      15  820.44    26.4  807.96    44.4  792.63
      55  785.35    62.7  781.33    71.6  777.87      76  775.18    84.8  768.18
    89.2  765.64   104.6  760.25   137.6  758.85   151.1  759.08   158.7  760.29
   168.8  763.83   182.7  764.78   190.9  767.46   194.7  767.97   226.3  766.23
   261.7  766.32   350.1  768.75   420.5  769.28   441.8  770.52   450.9  773.15
   459.7  776.79   477.1  781.88   487.4  786.53   499.6  792.93   519.5  806.69
#Mann= 5, -1 ,  0
       0     0.1       0   104.6   0.045       0   158.7     0.1       0
     180    0.06       0     290     0.1       0
Bank Sta=104.6,158.7
XS Rating Curve= 0 ,0
Exp/Cntr(USF)=0,0
Exp/Cntr=0.3,0.1

Type RM Length L Ch R = 1 ,20809   ,406.7,418.5,445.6
XS GIS Cut Line= 3
 1605733.9941416432753.9263047831605910.84969238432994.028211484
1606039.68486183433159.171474142
#Sta/Elev= 30
       0  794.56     3.6  793.92     8.2   790.8    18.1  777.03    28.1  769.18
      38  760.07      44  756.86    53.4755.1575    64.3  754.19    83.5   754.1
   96.92  755.17   106.4  758.22   111.5  758.69   123.5  755.92   127.4  755.83
   131.7  757.14   137.8  760.72   140.7     761   177.1  760.04   189.3  760.93
   251.6  762.21   316.6  766.33   377.5   771.4   418.1  776.48   443.4   783.8
   453.6  787.55   469.3  791.12   486.1  791.76   495.4  794.39   507.7  795.29
#Mann= 5, -1 ,  0
       0     0.1       0    53.4   0.045       0   96.92     0.1       0
     170    0.06       0     180     0.1       0
#XS Ineff= 2 , 0
                          170.73           764.8
Permanent Ineff=
       F       F
Bank Sta=53.4,96.92
XS Rating Curve= 0 ,0
Exp/Cntr(USF)=0,0
Exp/Cntr=0.3,0.1

Type RM Length L Ch R = 1 ,20391   ,638.1,631.3,633.1
XS GIS Cut Line= 4
1605732.29574024432667.9945161831605587.50124184432838.574336219
1605373.28472366433044.8569092861605224.52325269433110.311956509
#Sta/Elev= 30
       0  810.68    26.9  792.95    49.7  781.17    65.8  775.45    86.8  764.66
    99.2  761.18   267.1  758.43   315.2  753.68   332.2  755.31     365  754.48
   389.3750.6583   399.6  749.97   417.3  750.63   439.5  756.54   450.6  761.36
   461.7  762.18   493.5  769.82   522.4  780.38   527.9     784     553  809.81
   574.9  826.38     588  838.27   597.7  844.04   605.4  850.47   618.6   864.9
   627.3  878.52     636  888.66   653.5  892.03   673.5  899.52   683.7   901.2
#Mann= 5, -1 ,  0
       0     0.1       0   389.3   0.045       0   417.3     0.1       0
  423.75    0.06       0  551.14     0.1       0
Bank Sta=389.3,417.3
XS Rating Curve= 0 ,0
Exp/Cntr(USF)=0,0
Exp/Cntr=0.3,0.1

Type RM Length L Ch R = 1 ,19760   ,649.9,617.4,600.3
XS GIS Cut Line= 4
1605427.62570221432224.8158461131605376.87245364432321.116881863
1605078.85978895 432619.129546551605095.77753848432773.992022958
#Sta/Elev= 30
       0  826.47     7.5  821.22    14.2  817.74    17.2  814.88    20.2   811.6
    31.3  796.34    33.3   794.7    50.4  783.49      63  776.69    93.3  764.17
   113.7  758.53   177.8   749.2   189.8745.2568   198.5  744.79   228.7  745.28
   250.4  745.99   258.9  750.44   262.7  751.35   407.9  748.45   431.4  747.04
   477.6  749.95   563.9  751.93   584.7  753.65   592.1  755.43   608.2  761.92
   620.2  765.18   636.3  765.73   652.4  771.66   676.6  774.18   686.1  776.58
#Mann= 4, -1 ,  0
       0     0.1       0   189.8   0.045       0   228.7    0.06       0
  438.86     0.1       0
#XS Ineff= 2 , 0
                          262.19          787.63
Permanent Ineff=
       F       F
Bank Sta=189.8,228.7
XS Rating Curve= 0 ,0
Exp/Cntr(USF)=0,0
Exp/Cntr=0.3,0.1

Type RM Length L Ch R = 1 ,19142   ,497.9,486.7,471.4
XS GIS Cut Line= 4
1604714.64675274432398.6882310631604793.19280941432473.664012427
1604934.21868388432680.7399800061605005.62418994432809.269890917
#Sta/Elev= 30
       0  863.05     8.5  848.48    13.1  841.77    25.9  827.91    37.4  812.49
    61.8  790.59    68.4  782.97    79.4  772.58      96  762.56   104.2  759.11
   115.6  755.99   138.7  752.13   142.2  750.55   150.8  744.14   155.6  742.46
   218.5  742.03   237.9  739.81   256.7  738.54   277.9739.8256   286.3  745.57
   288.4  745.76   372.6  747.99   390.9   749.6   418.4  758.44   432.1  761.45
   441.3  762.41   451.6  760.82   468.7  764.43   494.8  772.69   506.2  778.92
#Mann= 4, -1 ,  0
       0     0.1       0  138.59    0.06       0   237.9   0.045       0
   277.9     0.1       0
Bank Sta=237.9,277.9
XS Rating Curve= 0 ,0
Exp/Cntr(USF)=0,0
Exp/Cntr=0.3,0.1

Type RM Length L Ch R = 1 ,18656   ,236.3,235.4,234.2
XS GIS Cut Line= 3
1604430.80986614432843.1875062971604750.34950577432928.874113571
1604869.95372842433003.849894936
#Sta/Elev= 30
       0  794.49     9.6  789.05    30.3  782.24    41.4  777.51    63.5  764.15
    84.2  757.12    88.3  754.24   100.7  738.97   104.9  734.99     109  733.87
   125.6  733.69   142.2  734.89   158.7  738.03   175.2  739.44   201.4  738.48
   237.4  740.44     254  742.49   299.5  742.73   305.9  744.08   320.2  750.26
   337.7  754.39   351.8     754   361.2   756.7   375.4  758.28   389.9   764.5
   417.9  772.89   432.1     780   446.2  790.49   462.4  807.33     472  815.83
#Mann= 5, -1 ,  0
       0     0.1       0      40    0.06       0   104.9   0.045       0
   142.2    0.06       0     170     0.1       0
Bank Sta=104.9,142.2
XS Rating Curve= 0 ,0
Exp/Cntr(USF)=0,0
Exp/Cntr=0.3,0.1

Type RM Length L Ch R = 1 ,18420   ,386.4,374.5,368
XS GIS Cut Line= 4
1604344.40769358433060.1557426191604430.35876569433091.009973633
1604655.15387737433135.0874465111604738.90107583433176.961045744
#Sta/Elev= 30
       0  782.65     8.2  779.78    29.4  774.66    46.4  767.56    80.4  757.09
   109.4   751.5   129.8   743.5   133.9  741.42     142  736.06   146.9734.1004
   154.3  733.08   186.9  732.93     195  733.02   199.1  734.11   203.2   736.1
   211.3  737.56   244.1   736.6   256.2  738.09   280.6  739.48   288.8  741.59
   305.4   747.7   325.9  756.77   348.3  768.14   361.7  772.04   370.7  776.64
   381.8  785.47   387.8  791.14     402  806.88   406.4  813.02     414   822.1
#Mann= 5, -1 ,  0
       0     0.1       0  131.32    0.06       0   146.9   0.045       0
   199.1    0.06       0  231.32     0.1       0
Bank Sta=146.9,199.1
XS Rating Curve= 0 ,0
Exp/Cntr(USF)=0,0
Exp/Cntr=0.3,0.1

Type RM Length L Ch R = 1 ,18046   ,296.8,277.7,263.7
XS GIS Cut Line= 3
1604313.45649213433529.4375769781604671.73361879433450.713006545
1604798.65690582433357.528821135
#Sta/Elev= 30
       0  817.86    10.9  803.43    19.1  794.94    35.5  782.75    51.9   777.8
    68.2  769.35    76.9  767.88   113.8  755.68   127.2   753.3   137.9   749.3
   162.4  743.57   174.7  737.59   191.1  736.45   203.4   730.6   211.6  728.34
   227.9  727.56   244.7  728.34   264.8  732.78   297.6  733.32   301.7  734.18
   330.4  745.98   342.6  749.37   367.3  758.27   397.5  761.21   417.3  762.01
   425.9  763.56   457.4  774.16     486  785.67   507.8  798.98   524.3  810.64
#Mann= 5, -1 ,  0
       0     0.1       0     160    0.06       0   211.6   0.045       0
   244.7    0.06       0     260     0.1       0
Bank Sta=211.6,244.7
XS Rating Curve= 0 ,0
Exp/Cntr(USF)=0,0
Exp/Cntr=0.3,0.1

Type RM Length L Ch R = 1 ,17768   ,427.7,405.2,391.2
XS GIS Cut Line= 4
1604583.70078698433869.9632632741604644.75249467433781.598949523
 1604794.1685161433543.8186143371604808.62813108433468.307291677
#Sta/Elev= 30
       0  859.27     1.7  858.82     6.6  855.13    16.3  845.22      26   837.2
    30.9   834.2    45.5  828.91      50  826.36    60.1  818.42    85.2  800.76
    90.5  794.94    99.2  778.43   116.4  768.53   141.7  752.21   162.8  735.05
   174.8  727.88   179.5  726.62   188.9   725.5   217.3  725.38   231.5  726.61
   241.5  729.74   264.4  730.44     276  732.18   297.6  730.93     326  733.18
   368.5  732.93   382.7  734.78   389.3  737.02   423.5  754.73   465.1  770.68
#Mann= 5, -1 ,  0
       0     0.1       0   127.4    0.06       0   179.5   0.045       0
   231.5    0.06       0   237.4     0.1       0
Bank Sta=179.5,231.5
XS Rating Curve= 0 ,0
Exp/Cntr(USF)=0,0
Exp/Cntr=0.3,0.1

Type RM Length L Ch R = 1 ,17363   ,299.8,305.5,313.2
XS GIS Cut Line= 3
  1604976.169024433980.5750284611605037.22073168433824.732511482
1605075.77970496 433464.84876093
#Sta/Elev= 30
       0  839.51     8.6  834.01    25.8  825.88      43  806.34    47.3   800.9
    55.9  787.08    60.2  783.43    89.5  773.72   107.4  765.79   124.6  760.78
   132.7  756.43   141.8  749.53   154.3  744.18   199.8  734.38   211.8  729.06
   335.5  727.38   348.6  724.53   376.8  723.84   384.6  722.42   392.9  721.94
   412.1  722.52     421  726.86     425  731.28   433.1   743.2   441.1  756.98
   449.2  766.67   460.9   777.5   473.3  792.96   513.5   820.7   529.3  829.42
#Mann= 5, -1 ,  0
       0     0.1       0  227.37    0.06       0  327.37     0.1       0
   384.6   0.045       0   412.1     0.1       0
Bank Sta=384.6,412.1
XS Rating Curve= 0 ,0
Exp/Cntr(USF)=0,0
Exp/Cntr=0.3,0.1

Type RM Length L Ch R = 1 ,17057   ,313.8,333.8,361.8
XS GIS Cut Line= 4
1605178.36816214433908.0950531081605248.64189093433849.533612449
1605383.33320445433651.595943022 1605440.7234163 433566.09623966
#Sta/Elev= 30
       0  741.04     7.5   737.4    17.9  729.65    23.1  728.41    38.7  731.06
    46.4  729.83      68  728.47    92.7  725.86   126.4  725.36   155.2  723.27
   174.9  723.87   181.1  722.51   188.1  718.44   192.6  717.33     207  717.21
   218.5  718.53     233  719.94   247.5  720.01   264.6   721.2   270.3  722.01
   273.2  723.26     291  736.76   305.6  746.54   339.4  773.98     351  786.17
   368.2  809.86   373.1  814.54   392.4  826.65   411.7  835.58   433.9  849.82
#Mann= 5, -1 ,  0
       0     0.1       0   91.48    0.06       0   188.1   0.045       0
   218.5    0.06       0  311.48     0.1       0
#XS Ineff= 2 , 0
          172.18  733.12
Permanent Ineff=
       F       F
Bank Sta=188.1,218.5
XS Rating Curve= 0 ,0
Exp/Cntr(USF)=0,0
Exp/Cntr=0.3,0.1

Type RM Length L Ch R = 1 ,16723   ,238.9,240,243.2
XS GIS Cut Line= 4
1605162.85674186 433981.219457441605291.78335003433955.434135806
1605517.90078589434038.7405595451605658.72831173434044.691018383
#Sta/Elev= 30
       0  757.95    25.8  744.79    42.1  738.45    54.3  730.65    58.4  729.31
    66.2   729.3    82.9  732.03   136.1  731.45   148.9  729.69   170.2  723.86
   229.9   718.4   244.7  715.63   251.2  714.43   272.5  714.16   282.1  714.47
   286.5715.5497   293.8  719.42   306.6  723.09   327.9  731.65   336.4  735.88
   366.3  743.18   382.7  743.98   410.7  751.92   438.7  757.06   454.7  763.19
   470.8  765.48   482.8  773.56   486.8  775.34   498.8  778.07   513.4  785.86
#Mann= 5, -1 ,  0
       0     0.1       0  171.48    0.06       0  191.48     0.1       0
   244.7   0.045       0   286.5     0.1       0
Bank Sta=244.7,286.5
XS Rating Curve= 0 ,0
Exp/Cntr(USF)=0,0
Exp/Cntr=0.3,0.1

Type RM Length L Ch R = 1 ,16483   ,230.8,229.7,229.7
XS GIS Cut Line= 4
1605155.29487893434154.3293880871605222.77308216 434175.21549861
1605423.60106796434271.6129317931605545.70448332434324.631520044
#Sta/Elev= 30
       0  756.08    21.8  742.77    30.2  739.08    53.6  730.97    76.6  725.66
    85.4  722.68    89.9  721.85   125.4  717.57   138.4  717.29   144.6  713.52
   147.6  711.97   162.6  711.47   169.7  711.82   177.3713.5475     183  714.04
   204.5  712.48   212.3  712.78   214.1  713.16   222.5  718.66   225.5  719.45
   258.4  724.67   282.5  727.18     294  729.06   312.7   733.5   337.1  741.21
   346.3   741.8   359.4  744.16   379.6  750.02     403  763.05   426.5  772.77
#Mann= 7, -1 ,  0
       0     0.1       0  100.64    0.06       0   144.6   0.045       0
   177.3    0.06       0  210.64     0.1       0  280.64    0.06       0
   323.4     0.1       0
Bank Sta=144.6,177.3
XS Rating Curve= 0 ,0
Exp/Cntr(USF)=0,0
Exp/Cntr=0.3,0.1

Type RM Length L Ch R = 1 ,16254   ,214.2,216,218
XS GIS Cut Line= 2
1605042.83120688434350.3375022261605389.86196634434502.966771433
#Sta/Elev= 30
       0  785.48    35.3  771.98    40.7  769.06    45.1  765.05    53.8  755.02
    66.9  741.79    84.4  726.57    88.8  724.13   104.8  718.61     115  716.49
   136.9  715.59   154.3  713.94   166.5  715.55   171.8  715.54   176.2  713.98
   181.7  710.85   184.7  710.13   187.8  710.08     209  710.27   215.1  710.88
   228.6  713.59   233.3  713.93   241.7  715.57   246.1  716.97   263.4  725.23
   272.3  728.11   287.9  731.47   298.5  732.83     316  734.16   379.1  738.19
#Mann= 6, -1 ,  0
       0     0.1       0   181.7   0.045       0   215.1     0.1       0
     230    0.07       0     280    0.06       0     340     0.1       0
Bank Sta=181.7,215.1
XS Rating Curve= 0 ,0
Exp/Cntr(USF)=0,0
Exp/Cntr=0.3,0.1

Type RM Length L Ch R = 1 ,16038   ,370.1,368.8,366.7
XS GIS Cut Line= 4
1604964.51279451434541.5373737831605024.37560052434561.057854003
1605154.51213532434637.838409534 1605259.9227285434644.345236274
#Sta/Elev= 30
       0   771.8    12.2  761.87    33.2     747    37.4  743.47    43.3  739.28
    49.7   735.6    54.3  733.54    62.7  730.23    71.2  727.46    76.6  725.11
    90.5  716.99    99.8  714.57     115  712.47   120.8  711.33   123.7  711.18
   132.3  712.83     137  712.84   144.2  711.98   158.8  709.12   164.8  708.46
   176.3  708.32   185.1   708.6   188.5709.1169   192.7  711.89   197.3  716.31
     202   719.2   203.6  719.64   255.7  727.19   299.8  730.92   319.7  731.65
#Mann= 5, -1 ,  0
       0     0.1       0  102.97    0.06       0   158.8   0.045       0
   188.5    0.06       0  314.06     0.1       0
Bank Sta=158.8,188.5
XS Rating Curve= 0 ,0
Exp/Cntr(USF)=0,0
Exp/Cntr=0.3,0.1

Type RM Length L Ch R = 1 ,15669   ,251.3,254.5,256.7
XS GIS Cut Line= 2
1604810.94704188434871.3703689431605097.24741844435000.060942243
#Sta/Elev= 30
       0  805.41     2.8   802.3     5.7   799.8    23.2   789.3      29  786.74
    41.9  782.46    49.5  779.27    53.9  777.05    58.3   774.1    61.4  770.17
    67.1  761.85    71.4  754.94    75.8  749.17    84.6  739.39      89  734.77
    92.5  731.61   101.6     724   110.9  717.35   119.7  712.45   122.8  711.09
   132.8  708.14   139.4  706.98     146  706.64   189.9  707.16     198  708.14
   210.5   712.6   216.2  715.47   220.6  716.59     268  718.78   313.9  719.44
#Mann= 4, -1 ,  0
       0     0.1       0   132.8   0.045       0     198     0.1       0
     200    0.06       0
Bank Sta=132.8,198
XS Rating Curve= 0 ,0
Exp/Cntr(USF)=0,0
Exp/Cntr=0.3,0.1

Type RM Length L Ch R = 1 ,15414   ,221.3,219.9,218.8
XS GIS Cut Line= 2
1604690.93223757435076.6969016231604983.01646012435237.198627874
#Sta/Elev= 30
       0  795.32    16.3  791.41    33.2  786.64    51.6  779.52    60.7  776.36
    69.8  772.35    83.5  763.27    88.1  760.04    92.1  756.82   109.7  737.26
   112.7  734.72   115.6  732.76     120  730.49   124.6  727.52   130.4  722.15
   136.2  715.32   142.8  708.21   147.4  705.63     153704.4121   157.5  703.85
   165.7  703.66   188.5  703.67   195.2  704.36   198.1  705.12   207.3  709.12
   215.8  711.89     225  713.11   270.6  714.67   304.1  715.13   333.3  715.16
#Mann= 4, -1 ,  0
       0     0.1       0      80    0.06       0     153   0.045       0
   195.2    0.05       0
Bank Sta=153,195.2
XS Rating Curve= 0 ,0
Exp/Cntr(USF)=0,0
Exp/Cntr=0.3,0.1

Type RM Length L Ch R = 1 ,15194   ,240.1,249.5,255.4
XS GIS Cut Line= 2
 1604607.0664707 435290.699203291604894.81280875435428.065545577
#Sta/Elev= 30
       0  751.69      10  749.99    32.2   745.4    41.1  742.56      60  734.81
    69.3  729.53    78.5  723.45    86.2  719.03    89.2  717.05    94.2  713.09
    95.2  712.54    98.7  711.11   107.2  710.87     112  711.31   116.2  710.85
   119.2  708.87   125.3  703.79   129.7   702.9   143.5  702.36   165.2  702.75
   169.6  702.99     174  703.75   182.9  706.06   196.2  709.05   213.9  711.22
   218.3  711.41   227.2  711.22   240.5  712.09   302.6   713.8   318.9  714.76
#Mann= 4, -1 ,  0
       0     0.1       0      60    0.06       0   125.3   0.045       0
     174    0.05       0
Bank Sta=125.3,174
XS Rating Curve= 0 ,0
Exp/Cntr(USF)=0,0
Exp/Cntr=0.3,0.1

Type RM Length L Ch R = 1 ,14945   ,289.4,300.1,308.8
XS GIS Cut Line= 3
 1604540.5522418435452.6468910381604701.05396805 435663.75726971
1604722.27408787435722.510663682
#Sta/Elev= 30
       0   709.8    14.9  708.88    32.3  709.27    45.1  710.29    65.4  709.77
    78.6  707.55    85.3  707.03   100.4  704.91   105.4  704.47   116.6  704.55
   124.9  702.44   130.9  699.98   135.5  699.32   145.6  699.22   162.3     700
   170.7  701.01   175.7  702.78   185.8  712.23   190.8   715.7   195.8  716.41
   210.9  716.61     224  721.98     231  725.34     236  727.14   251.1  730.69
     266   732.6     283  736.46   304.3  743.42   317.1  748.31   327.7  751.18
#Mann= 6, -1 ,  0
       0    0.06       0     120    0.05       0   130.9   0.045       0
   162.3    0.05       0     200    0.07       0     240    0.06       0
Bank Sta=130.9,162.3
XS Rating Curve= 0 ,0
Exp/Cntr(USF)=0,0
Exp/Cntr=0.3,0.1

Type RM Length L Ch R = 1 ,14645   ,522.1,526.1,529.7
XS GIS Cut Line= 3
1604331.45070321435450.5320702151604356.17664482435742.037908161
1604366.58756761435830.530751824
#Sta/Elev= 30
       0   721.2    22.1  712.54    34.1  710.82    46.2   707.7    66.2  706.57
   154.6  704.22   166.6  702.77   178.6  702.38   188.9700.0169   198.7  698.28
   210.8  697.88   222.8  698.11   226.8  698.86   228.2  699.93   230.8  701.81
   234.8  707.02   238.3  709.85   246.7  714.78   254.9  717.34     275  718.62
     279  719.81   291.1  726.46   311.2  734.44   323.6  740.82   335.3  745.71
   339.4   748.4   343.4  752.33   359.4  769.63   371.6  783.94   381.7   792.9
#Mann= 5, -1 ,  0
       0    0.06       0     100    0.05       0   188.9   0.045       0
   228.2    0.06       0  292.55     0.1       0
#XS Ineff= 2 , 0
           79.84  717.38
Permanent Ineff=
       F       F
Bank Sta=188.9,228.2
XS Rating Curve= 0 ,0
Exp/Cntr(USF)=0,0
Exp/Cntr=0.3,0.1

Type RM Length L Ch R = 1 ,14119   ,259.7,257.2,254.4
XS GIS Cut Line= 4
1603848.33150469435418.8178789981603839.22194725435517.721645444
1603861.34515817435741.5564852961603879.56427304435785.802907127
#Sta/Elev= 30
       0  740.74    13.8  737.78    45.9  728.56      62  724.54      78  721.38
    94.1   718.9    98.1  717.71   102.2  715.37   106.4  712.48   110.2  709.55
   118.2  702.58   126.3  696.19   130.3  694.02   134.3  694.16     143  696.17
   154.4  699.04   158.4  699.45   190.6  700.94   258.9  702.71   263.7  702.64
     271  701.72   285.6  702.87   311.2  703.57   318.5  704.52   331.5  705.45
     344  707.28   349.1  708.32   352.5  709.67   359.3  711.34   372.1  711.75
#Mann= 6, -1 ,  0
       0     0.1       0   126.3   0.045       0     143     0.1       0
  229.32    0.05       0  324.25    0.07       0  354.25    0.06       0
Bank Sta=126.3,143
XS Rating Curve= 0 ,0
Exp/Cntr(USF)=0,0
Exp/Cntr=0.3,0.1

Type RM Length L Ch R = 1 ,13861   ,352.4,347.4,343.2
XS GIS Cut Line= 3
1603555.52430139435478.6806850051603649.22260645435796.213829911
1603709.08541245435891.213500313
#Sta/Elev= 30
       0  755.95    14.9  751.76    39.5  746.14    47.8  743.33    56.2  739.33
    64.5  733.36    68.7  728.84    72.8  723.46    81.2  715.65    86.9  709.84
    89.5  706.83    93.7  701.18    97.9   697.4     102  694.57   106.2  693.33
   117.9  692.19   127.1  692.06   139.6   692.2   147.9  693.38   156.2  696.23
   202.1     698     223  699.82   281.4   700.7     359  706.07     374  707.81
   383.5  710.41   407.1  710.36   416.6  711.91   435.5  713.69   443.4   715.2
#Mann= 7, -1 ,  0
       0     0.1       0   106.2   0.045       0   147.9     0.1       0
     180    0.06       0     280    0.05       0  381.07    0.07       0
  391.07    0.05       0
Bank Sta=106.2,147.9
XS Rating Curve= 0 ,0
Exp/Cntr(USF)=0,0
Exp/Cntr=0.3,0.1

Type RM Length L Ch R = 1 ,13514   ,383.8,372.8,362.1
XS GIS Cut Line= 3
1603205.61620668435623.4944091421603410.94273937435925.700362172
1603486.13273725436009.566129041
#Sta/Elev= 30
       0  751.23    25.8   741.7    35.1  737.29    39.9  734.16    47.2   726.3
    64.1  705.79    68.5  701.34    73.8  696.84    78.6   691.8    81.9690.0233
    83.5  689.52   104.1  689.26   111.2  690.01   120.6   691.4   141.5  691.33
   151.2  693.22   163.8  694.66   186.8  696.45     214  697.02   272.1  695.77
   310.7  696.38   339.8   697.9   359.1  699.56   393.7  700.98   406.8  704.18
   428.3  703.21     433   704.3     439   706.5   461.7  708.84     478  713.62
#Mann= 6, -1 ,  0
       0     0.1       0    81.9   0.045       0   111.2     0.1       0
     150    0.05       0  385.36    0.07       0  465.36    0.06       0
Bank Sta=81.9,111.2
XS Rating Curve= 0 ,0
Exp/Cntr(USF)=0,0
Exp/Cntr=0.3,0.1

Type RM Length L Ch R = 1 ,13141   ,230.5,229.3,227.8
XS GIS Cut Line= 4
1602976.61060177435967.0611470721603006.02015727 435997.41939791
1603207.14356907436057.1872042461603341.86981317436137.276860119
#Sta/Elev= 30
       0  754.73     7.6  750.23    33.8   737.3      57   722.8    69.5  712.26
    73.7   708.1      82   694.2    86.2   690.4    90.4  688.28    94.5  687.21
   104.4  686.29   110.8  685.68   132.1  685.26   136.3  685.34   141.7  686.28
   152.9  689.59   157.1  690.09   169.6  691.18   190.5  691.45   211.4  693.89
   236.4  695.44   281.1  694.89   313.6  695.44   325.3  696.11     337  698.91
   345.7  698.94   360.2  698.06   369.5  701.54   392.4  704.87   408.8  708.42
#Mann= 6, -1 ,  0
       0     0.1       0   104.4   0.045       0   141.7     0.1       0
  182.27    0.05       0  232.27    0.06       0  408.82     0.1       0
Bank Sta=104.4,141.7
XS Rating Curve= 0 ,0
Exp/Cntr(USF)=0,0
Exp/Cntr=0.3,0.1

Type RM Length L Ch R = 1 ,12912   ,309.9,309.7,310.2
XS GIS Cut Line= 4
1602940.77147097436179.2648844731602958.69127181436227.753757338
1603227.48828444 436285.72958359 1603299.1674878436325.785609001
#Sta/Elev= 30
       0   726.2     9.9  724.63    21.2  721.72    44.3  713.94    51.7  710.43
    53.1  710.38    57.2  708.79    65.4  703.75    77.1  695.28    83.8  691.15
    85.9  690.17    94.1  688.13   102.3  684.93   106.3  684.43   114.5  683.75
     135  683.94   139.1  684.41   159.5  688.95     180   689.6   208.4  693.24
   235.3  691.38   255.5  691.24   274.1  691.89   290.5   694.3   329.2  708.14
   346.8  715.81     364  726.19   373.4  731.27   396.1  746.41   408.8  752.87
#Mann= 5, -1 ,  0
       0     0.1       0   106.3   0.045       0   139.1     0.1       0
  181.69    0.07       0  281.69     0.1       0
#XS Ineff= 2 , 0
                          209.56          720.83
Permanent Ineff=
       F       F
Bank Sta=106.3,139.1
XS Rating Curve= 0 ,0
Exp/Cntr(USF)=0,0
Exp/Cntr=0.3,0.1

Type RM Length L Ch R = 1 ,12602   ,205.9,207.1,208.4
XS GIS Cut Line= 4
 1602825.5497077436478.1615136211602845.46059752436519.154522083
1603085.56250422436571.859818676 1603172.2334364436596.455623753
#Sta/Elev= 30
       0  692.15     3.7  691.24    11.5  690.55    56.5  689.55    72.9  689.68
   119.5  687.32   150.7  686.97     163  684.95   171.1  682.18   175.2  681.46
   183.4  681.06   199.8  681.13   203.9  681.42   205.6682.1586     208  683.26
   212.1  686.41   216.2  687.79   232.6  688.34   240.8  687.27   244.9  687.94
   250.4  689.98     274  691.34   281.7  692.61   297.2  701.09   323.1  712.68
   335.6  719.78   343.9  723.42   360.6  732.61   367.1  734.71   381.5  737.97
#Mann= 4, -1 ,  0
       0     0.1       0   171.1   0.045       0   205.6    0.07       0
  291.39     0.1       0
#XS Ineff= 2 , 0
                          228.99          695.57
Permanent Ineff=
       F       F
Bank Sta=171.1,205.6
XS Rating Curve= 0 ,0
Exp/Cntr(USF)=0,0
Exp/Cntr=0.3,0.1

Type RM Length L Ch R = 1 ,12395   ,399.4,409.5,423
XS GIS Cut Line= 4
1602756.73054319436662.0017616071602790.46193301436707.328316677
1603012.87828463436773.7369903841603070.85411088436810.630697999
#Sta/Elev= 30
       0  688.53    13.1  688.72    24.2  688.26      53  688.03   120.8  685.99
   158.5  685.56   170.9  685.17   183.5  684.15   187.4  683.53   194.9  680.41
     196  679.99   200.2  679.47     221   679.2   225.2  679.26   229.2  680.41
   233.6  684.02   237.7  688.24   241.9   690.5   246.1  691.05   254.4   691.6
   266.9  691.56     271  692.61   283.6  698.11   288.6  699.77   298.8  704.62
   307.5   709.1   320.9  717.37   342.2  726.78   353.4  731.07   357.3   732.3
#Mann= 6, -1 ,  0
       0    0.05       0    56.5     0.1       0   156.5    0.07       0
   194.9   0.045       0   229.2    0.07       0   266.5     0.1       0
Bank Sta=194.9,229.2
XS Rating Curve= 0 ,0
Exp/Cntr(USF)=0,0
Exp/Cntr=0.3,0.1

Type RM Length L Ch R = 1 ,11986   ,394.9,403.6,417.5
XS GIS Cut Line= 4
1602496.85109644436745.247300251 1602525.7703264436799.872512388
1602757.12416604437156.543015167 1602773.1904049437232.054337827
#Sta/Elev= 30
       0  694.28     8.2  690.77    21.8  686.51    39.9  684.79   104.5  684.09
   134.1  682.33   186.6  682.36   240.4  683.57   280.9  685.39   312.7  679.78
   356.1  680.83     386677.1945   410.6  676.62   418.9  677.19   422.6  679.05
     425  681.04   433.6  693.93   439.9  698.75     444  699.99   477.4  703.76
   480.4  704.65   482.2  705.31     491  713.62   495.1  716.67   499.2     719
   503.3  720.15   515.6  721.37   548.3  726.24   556.9   726.4   564.1  727.38
#Mann= 5, -1 ,  0
       0     0.1       0  371.81    0.07       0     386   0.045       0
   418.9    0.07       0  556.94    0.05       0
#XS Ineff= 2 , 0
          275.63   712.6
Permanent Ineff=
       F       F
Bank Sta=386,418.9
XS Rating Curve= 0 ,0
Exp/Cntr(USF)=0,0
Exp/Cntr=0.3,0.1

Type RM Length L Ch R = 1 ,11582   ,478.7,476.2,469.5
XS GIS Cut Line= 4
1602278.35024789436897.8765694581602331.36883614436995.880626527
1602292.80986287 437293.106045511602341.00857946437424.849204194
#Sta/Elev= 30
       0  689.25    26.9   686.1    75.8  683.06   160.5  683.41   168.6  682.13
   176.6  679.41   184.7  677.84   200.8  676.89   212.9  674.68   230.2673.7051
   241.2  673.26   261.3  673.69   277.5   677.7   289.9  679.34   309.7  680.48
     342  680.54   354.1  681.96   362.2  684.36   382.3  692.02   394.4  695.24
   413.3  699.17   428.9   703.4   447.6  710.42   470.2  716.51   488.1  722.21
   508.5  730.11   512.8  731.29   525.5  732.41   534.9  735.75   551.4  737.13
#Mann= 6, -1 ,  0
       0     0.1       0   230.2   0.045       0   261.3    0.07       0
  341.43     0.1       0  401.43    0.05       0  421.14     0.1       0
#XS Ineff= 2 , 0
                          311.86          711.32
Permanent Ineff=
       F       F
Bank Sta=230.2,261.3
XS Rating Curve= 0 ,0
Exp/Cntr(USF)=0,0
Exp/Cntr=0.3,0.1

Type RM Length L Ch R = 1 ,11106   ,430.2,431.1,432.6
XS GIS Cut Line= 4
1601885.87781777436951.7568723031601857.31561535437032.088066623
1601900.15891898437301.643852006 1601921.5805708437458.735965342
#Sta/Elev= 30
       0  776.97    30.2  759.89    45.8  752.38    64.5  745.31    93.8  732.41
     106  728.53   118.1  725.79   126.2  722.41   130.3  719.98     137  714.38
     144  706.65   150.5  698.75   154.6  692.85   158.6     685   166.7  673.61
   170.8  670.64     191     670   207.2   669.4   229.3670.0423   239.6  674.15
     272  676.02   292.3  675.38   312.5  677.89   369.2   680.6   405.5  684.26
   409.6  685.22   437.8  696.67   470.1  706.53   494.3  712.21   516.7  716.44
#Mann= 5, -1 ,  0
       0     0.1       0     191   0.045       0   229.3     0.1       0
  275.26    0.07       0   378.2    0.05       0
#XS Ineff= 2 , 0
                          270.88          726.04
Permanent Ineff=
       F       F
Bank Sta=191,229.3
XS Rating Curve= 0 ,0
Exp/Cntr(USF)=0,0
Exp/Cntr=0.3,0.1

Type RM Length L Ch R = 1 ,10675   ,313.5,312.8,311.5
XS GIS Cut Line= 4
1601458.19409844436933.4426823231601434.98730897437015.559014294
1601472.47519965437442.2069130131601454.62382313 437565.38141097
#Sta/Elev= 30
       0  715.64    10.7  711.82    28.2  701.91    53.1  694.59      78  678.84
    86.3  676.63   110.4  673.91   134.5  672.58   242.9   673.1   283.1  670.31
   295.1  665.13   299.1   664.2   323.2     664   331.3  665.14   343.3  666.85
   355.3  670.68   391.5  670.24   419.6  672.84   435.7  669.97   439.7  670.49
     455  674.62   479.8   684.9   503.9  687.09   512.2  688.94     520  692.83
   544.3  708.29     576  736.77   592.8  747.79     613  767.07   638.1   792.7
#Mann= 4, -1 ,  0
       0     0.1       0   295.1   0.045       0   331.3    0.06       0
  395.33     0.1       0
#XS Ineff= 2 , 0
                          413.33          689.91
Permanent Ineff=
       F       F
Bank Sta=295.1,331.3
XS Rating Curve= 0 ,0
Exp/Cntr(USF)=0,0
Exp/Cntr=0.3,0.1

Type RM Length L Ch R = 1 ,10362   ,560.8,542.8,523.4
XS GIS Cut Line= 4
1601126.50870232437021.1636862141601128.29383998437158.619285383
1601167.56686831437440.6710343271601210.41017195437545.994155768
#Sta/Elev= 30
       0  678.39    23.4  676.26    55.4  674.09   147.5  669.59     204  667.76
   212.1   666.8   229.1  662.96   236.3  661.78   244.4  661.75   260.6  661.81
  267.42  662.97   280.8  665.69   300.9  667.26   309.2  668.37   329.2  672.98
   337.5  674.44   365.6  676.24   373.6  679.32   387.2  682.86   393.8   685.3
   401.9  689.67   430.7  703.07   443.7  708.04   453.3  713.25   465.3   721.3
   478.2  727.95   493.2  733.67   504.1  736.58   521.4  743.86   535.9  747.76
#Mann= 7, -1 ,  0
       0     0.1       0     100    0.06       0  197.47     0.1       0
   229.1   0.045       0  267.42     0.1       0  297.47    0.06       0
  397.47     0.1       0
#XS Ineff= 2 , 0
          191.76  676.91
Permanent Ineff=
       F       F
Bank Sta=229.1,267.42
XS Rating Curve= 0 ,0
Exp/Cntr(USF)=0,0
Exp/Cntr=0.3,0.1

Type RM Length L Ch R = 1 ,9819    ,148.9,137.5,128
XS GIS Cut Line= 4
1600475.93567455 437337.543788251600567.03124891 437382.36859468
1600770.91182009437534.194551944 1600896.7104704437606.492626832
#Sta/Elev= 30
       0  720.84     4.7  719.69    26.9  709.77    49.2  703.33    61.1  701.11
    84.9   698.7    89.4  696.76   102.9  687.93   111.9  684.12   131.9  677.99
   152.7  665.84  169.15  659.58   175.3  658.52   187.7  658.38   205.6  658.49
   218.2  659.56   235.3  660.54   266.8  663.68   281.1  663.18   292.4  663.68
   309.7  667.72   335.4  666.39   349.7  669.21   375.6  669.47   390.6  670.66
   398.6  672.23   435.5  683.74   458.6  686.97   467.8  689.27   500.8  694.43
#Mann= 5, -1 ,  0
       0     0.1       0  169.15   0.045       0   218.2     0.1       0
  301.53    0.06       0  415.73    0.05       0
Bank Sta=169.15,218.2
XS Rating Curve= 0 ,0
Exp/Cntr(USF)=0,0
Exp/Cntr=0.3,0.1

Type RM Length L Ch R = 1 ,9682    ,32.9,32.3,33.4
XS GIS Cut Line= 4
1600365.42564554437568.7846119271600439.16182596437538.102143216
1600747.80290388437591.9784888841600894.13748012437662.963951606
#Sta/Elev= 30
       0  688.26    24.6  678.92    76.6  678.41      89  675.89   113.3  673.84
   121.4  671.72     158  668.27   187.1  664.19   203.8  660.79  211.48  657.75
   214.8  657.05     227  656.63   240.4   656.8   251.4  657.76   263.6  657.92
   275.7   660.8     296  662.09   312.3  664.93   332.6  666.55   356.9  665.18
   366.3  666.25   424.6  668.23   429.1  669.14   438.7  672.69   453.7  677.32
   473.5  682.68   486.6  685.29   504.9  687.66   526.9  691.36   555.8  698.03
#Mann= 5, -1 ,  0
       0     0.1       0  211.48   0.045       0   251.4     0.1       0
  269.87    0.06       0  443.17    0.05       0
Bank Sta=211.48,251.4
XS Rating Curve= 0 ,0
Exp/Cntr(USF)=0,0
Exp/Cntr=0.3,0.1

Type RM Length L Ch R = 1 ,9649    ,170.1,166.9,164.2
XS GIS Cut Line= 4
1600363.81937845437600.9100261271600437.55555886437570.227557416
1600746.19663678437624.1039030851600892.53121302437695.089365806
#Sta/Elev= 30
       0  692.58       9  687.86    30.6  679.61      61  678.59    78.3   678.8
    82.5  678.41   106.8  673.46   163.1  667.63     174  666.97     184  668.14
     188  667.87   204.3   664.3   208.3  662.64  215.16  657.69   220.5  656.65
   232.7  656.31   257.1  657.71   277.4  657.83   289.5  662.38   293.6   663.3
   301.7  663.35     322  665.98   342.3  664.63   358.6  666.28   404.2  667.31
   417.5  668.29   430.9  673.59   453.1  679.68   510.9  690.09   555.8  700.43
#Mann= 5, -1 ,  0
       0     0.1       0  215.16   0.045       0   257.1     0.1       0
  269.87    0.06       0  369.87    0.05       0
Bank Sta=215.16,257.1
XS Rating Curve= 0 ,0
Exp/Cntr(USF)=0,0
Exp/Cntr=0.3,0.1

Type RM Length L Ch R = 1 ,9482    ,405.3,415.2,425.9
XS GIS Cut Line= 4
1600407.66264721437713.7525462021600498.70466744437751.240436884
1600670.07788199437770.8769510511600823.59972002437808.364841734
#Sta/Elev= 30
       0  693.12     4.8  691.86    13.5  688.35    30.1  679.37    48.1  668.86
    52.4  666.89    59.8  664.73    69.7   663.6   107.7  663.32   136.1   662.3
   156.2  658.98   168.3  655.56   191.8   655.1   204.6  654.29   212.6  654.51
  215.88   655.1   220.7  656.65   228.7  660.31   236.8  662.15   244.8  662.58
   260.9  662.51   285.4  666.78   293.6  667.53   333.6  668.01   338.9  668.48
     343  669.47   351.3   672.8   363.6  676.07   392.5  681.39     429  689.41
#Mann= 5, -1 ,  0
       0     0.1       0   191.8   0.045       0  215.88     0.1       0
  228.46    0.07       0  428.99    0.08       0
Bank Sta=191.8,215.88
XS Rating Curve= 0 ,0
Exp/Cntr(USF)=0,0
Exp/Cntr=0.3,0.1

Type RM Length L Ch R = 1 ,9067    ,399.4,403,406.9
XS GIS Cut Line= 3
1600236.75087288437907.3995478011600582.17500845438243.183940057
1600708.91978171438294.595904421
#Sta/Elev= 30
       0  742.59    70.5  713.27   105.1  694.29   116.3  685.49   124.8  675.54
     133  667.79   141.8  660.85   147.4  658.28   162.3  657.37   195.5   659.1
   222.3  658.19   236.9  659.34   254.1  655.87   288.9  657.52   305.9  656.62
   328.2  652.63   345.5  651.37   361.7  652.61   374.6  659.02   395.2  660.45
   410.5  662.98   469.9  663.04   501.1  665.16     514  667.41   522.7  664.85
   531.3  667.06   545.7  667.22     561  669.26   583.1  681.12   618.5  708.11
#Mann= 7, -1 ,  0
       0     0.1       0     290    0.06       0   328.2   0.045       0
   361.7    0.06       0     410    0.07       0     430    0.06       0
  531.74     0.1       0
#XS Ineff= 2 , 0
          237.53  695.03
Permanent Ineff=
       F       F
Bank Sta=328.2,361.7
XS Rating Curve= 0 ,0
Exp/Cntr(USF)=0,0
Exp/Cntr=0.3,0.1

Type RM Length L Ch R = 1 ,8664    ,483.4,480.8,485.8
XS GIS Cut Line= 3
 1600007.7994809438148.5410294581600261.28902742 438543.05645045
1600341.62022174 438669.80122371
#Sta/Elev= 30
       0  718.89    33.3  714.22      45  709.68    66.6  693.45    81.3  679.33
    90.3  672.06   110.2   657.6     116  654.46   156.9  651.88   215.2  652.33
   246.2648.8842     255  648.25   276.4648.8569   280.5  650.13   285.3  654.03
     290  655.52   337.6  655.74   422.4  659.36   451.8  662.16   470.7  662.55
     501  667.15   513.3  671.78     537   690.2   551.2  697.26   560.7  705.68
   570.1  718.48   574.9   723.7   579.6  726.05   603.3     732     619  739.47
#Mann= 6, -1 ,  0
       0     0.1       0   246.2   0.045       0   276.4     0.1       0
     410    0.07       0     420    0.06       0  538.93     0.1       0
Bank Sta=246.2,276.4
XS Rating Curve= 0 ,0
Exp/Cntr(USF)=0,0
Exp/Cntr=0.3,0.1

Type RM Length L Ch R = 1 ,8183    ,874,863,851.8
XS GIS Cut Line= 4
1599628.32672191 438242.308506761599635.46727251438320.854563428
  1599853.254066438758.2132880571599942.51094858438908.164850787
#Sta/Elev= 30
       0   700.1    18.3  695.36    42.4     687    70.5  680.51      97  666.97
   123.2  657.94   147.7  645.23   167.9     644     179645.1838   214.9  648.16
   234.2   647.6   284.1  650.47     449  649.78   489.6  654.06   498.6  657.49
   514.6  667.74   538.8  669.19   547.7  672.72   561.1  675.33   579.5  684.19
   594.6  688.17   611.9  697.02   627.8   703.3   649.3  717.23   667.5  723.39
   681.9  725.66   695.8  729.94   725.9  743.57   733.1  749.07     742  758.41
#Mann= 7, -1 ,  0
       0     0.1       0   147.7   0.045       0     179     0.1       0
  278.87    0.08       0  308.87    0.05       0  388.87    0.06       0
  528.87     0.1       0
Bank Sta=147.7,179
XS Rating Curve= 0 ,0
Exp/Cntr(USF)=0,0
Exp/Cntr=0.3,0.1

Type RM Length L Ch R = 1 ,7320    ,558.4,562.1,564.6
XS GIS Cut Line= 3
1598777.45079953438607.4695716851599338.21420448439089.873024847
1599465.54912612439114.360509779
#Sta/Elev= 30
       0  745.36    16.8  732.96      65  705.72   124.9  664.12   150.1  652.77
   167.2   647.9   177.6  639.08   179.5  638.33   209.3  637.42   230.4  638.38
   252.2  641.88     309  641.03   337.3  642.76   399.2  642.42   581.5  644.09
   601.1  645.07   620.9  650.63   631.4   656.5   635.2  657.48   646.5  658.35
   668.3  656.81     672  657.59   674.9  659.65   684.2  674.08   691.9  682.61
   715.8   694.4   767.5  711.98   794.9  718.62   844.7  732.82   869.4     741
#Mann= 5, -1 ,  0
       0     0.1       0   179.5   0.045       0   230.4     0.1       0
     620    0.07       0  749.71     0.1       0
#XS Ineff= 2 , 0
                          515.33          657.52
Permanent Ineff=
       F       F
Bank Sta=179.5,230.4
XS Rating Curve= 0 ,0
Exp/Cntr(USF)=0,0
Exp/Cntr=0.3,0.1

Type RM Length L Ch R = 1 ,6758    ,532.7,533.7,529.1
XS GIS Cut Line= 4
1598473.80598638439008.3297000231598506.86409103439072.242035696
1598923.39620973439587.9484683651598991.71629269439742.219623437
#Sta/Elev= 30
       0   761.7    19.7  749.05    67.8  712.51    73.9  705.67    84.4   690.7
    98.7  675.76   108.3  664.02   137.6  639.61   144.2     638   208.6633.6176
   236.9   632.5   249.4  633.61   258.6  637.13   272.9   637.5   308.9  644.84
   324.3  642.09     350  643.81   579.4  644.92   656.2  649.47   668.8  648.05
   679.1   649.5   689.3  652.14   729.6  671.47   766.1  685.96   779.3  690.03
   796.8  701.98   809.9  713.06   862.4  743.19   875.9  754.46   903.6  772.85
#Mann= 8, -1 ,  0
       0     0.1       0   208.6   0.045       0   249.4     0.1       0
  311.96    0.08       0  351.96     0.1       0  471.96    0.05       0
  601.96    0.07       0  731.96    0.05       0
Bank Sta=208.6,249.4
XS Rating Curve= 0 ,0
Exp/Cntr(USF)=0,0
Exp/Cntr=0.3,0.1

Type RM Length L Ch R = 1 ,6225    ,429.9,432.4,433
XS GIS Cut Line= 4
1597844.33540537439231.8541533671597980.37698833439298.363371701
1598503.38129614439812.298240645 1598663.6080494440026.941627087
#Sta/Elev= 30
       0  711.46    44.3  699.31     114  694.33   171.7  687.92   188.8  684.17
   207.1   673.4   237.6  648.48   260.3  638.12     381  635.75   407.3   631.3
   434.2  630.91   444.1  631.24   472.4  634.95   493.2  635.16   514.8  643.54
   543.6  648.51   661.4     645   797.7  646.05   818.4  656.24   873.6  691.12
     900  692.86   908.2  699.41   914.9  707.95   924.9  714.84   988.3  740.48
  1024.7  766.65  1039.7  774.69  1074.7   787.1  1114.6   794.8  1152.5  798.12
#Mann= 9, -1 ,  0
       0    0.05       0     120    0.06       0  271.43    0.05       0
   407.3   0.045       0   444.1    0.07       0  551.43    0.05       0
  701.43    0.06       0  841.43    0.08       0  974.68     0.1       0
Bank Sta=407.3,444.1
XS Rating Curve= 0 ,0
Exp/Cntr(USF)=0,0
Exp/Cntr=0.3,0.1

Type RM Length L Ch R = 1 ,5792    ,228.4,231.4,236.1
XS GIS Cut Line= 2
1597689.27462591439574.4295902961598139.84434867440078.871779901
#Sta/Elev= 30
       0  685.04    24.3  675.96    40.3  667.43      46  662.77    54.5  652.78
    65.8  643.13    76.3  636.68    82.3  635.24     114  632.08   214.4  634.24
     250  631.77   262.5  629.69   286.3629.8896   303.8   628.8   333.2629.8529
   335.4  630.81   340.6  636.24   343.5  637.09   371.8  639.93   421.2  641.85
   490.6  642.66   541.8  638.09   589.9  638.18   592.8  639.33   595.6  642.41
   609.7  660.19   623.9  673.14   632.4  679.46   646.4  687.34   676.4  696.61
#Mann= 9, -1 ,  0
       0    0.06       0      10     0.1       0   286.3   0.045       0
   333.2     0.1       0     410    0.05       0     420     0.1       0
     540    0.05       0     570    0.06       0     670     0.1       0
Bank Sta=286.3,333.2
XS Rating Curve= 0 ,0
Exp/Cntr(USF)=0,0
Exp/Cntr=0.3,0.1

Type RM Length L Ch R = 1 ,5561    ,67.8,65.3,62.8
XS GIS Cut Line= 5
1597692.71504931439629.645565609  1597649.900396439850.309980525
1597728.00964555439971.6375732821597736.75872478440166.330938898
1598048.77408062440206.386964308
#Sta/Elev= 30
       0  665.69       7  663.26    19.2  666.28    23.3  665.61    92.6  648.59
     113  646.79   141.5  640.65   153.7   640.3   186.3  635.85   210.7  635.36
   224.8   636.6   236.3  632.93     256  631.76     275  628.18   298.8  627.78
   317.5  628.19   327.3  628.39   354.5  633.34     394  632.84   465.8  636.17
   530.1  635.44     564   632.1   579.4  635.79   619.8   638.6   676.2  638.93
   781.1  635.68   789.2  638.69   801.2  649.59   821.4  663.32   878.5   670.8
#Mann= 10, -1 ,  0
       0     0.1       0     130    0.06       0     150     0.1       0
  254.78    0.08       0  264.78    0.07       0     275   0.045       0
   317.5    0.07       0  379.08    0.06       0  603.97    0.05       0
  703.97    0.06       0
#XS Ineff= 2 , 0
                          487.08          644.47
Permanent Ineff=
       F       F
Bank Sta=275,317.5
XS Rating Curve= 0 ,0
Exp/Cntr(USF)=0,0
Exp/Cntr=0.3,0.1

Type RM Length L Ch R = 1 ,5496    ,292.2,272.4,252.7
XS GIS Cut Line= 6
1597650.78326547439643.7251752871597615.02361332  439854.0042326
1597617.22311211439926.3110182121597671.29874641439990.822301242
1597685.10753412440202.1705405811598035.17121116440232.062195311
#Sta/Elev= 30
       0  678.76    41.4  672.76    53.6  669.37    73.9  666.13    98.2  663.69
   135.2  656.13   187.5  648.46   214.8  646.77   243.8     638   267.3  633.53
   286.4  631.75   294.9  628.29   326.2  627.59   346.1  628.25   365.9  629.95
   447.7  631.82   616.7  630.69   628.8  632.72   640.8  637.12   660.9  638.45
     677  637.74   737.2   630.9   801.4  636.77   833.5  635.89   837.5  636.51
   841.6  639.29   853.6  655.36   857.6  659.18   860.3  660.23     933  669.12
#Mann= 8, -1 ,  0
       0    0.06       0     140     0.1       0   243.3    0.08       0
   294.9   0.045       0   346.1    0.08       0  369.82    0.06       0
  671.61    0.05       0  771.61    0.06       0
#XS Ineff= 2 , 0
                          660.52          650.65
Permanent Ineff=
       F       F
Bank Sta=294.9,346.1
XS Rating Curve= 0 ,0
Exp/Cntr(USF)=0,0
Exp/Cntr=0.3,0.1

Type RM Length L Ch R = 1 ,5223    ,90.7,87.8,82.1
XS GIS Cut Line= 3
1597329.27974292440185.4243478251597413.14550979440194.100116812
1598023.34126185440249.046653727
#Sta/Elev= 30
       0  728.83    34.6  711.87    47.1  700.68    67.2  689.06    99.3  680.08
   111.4  675.53   143.5  668.23   175.7  654.82   207.8  646.22   218.2  638.09
   235.9   627.9     260  626.26   292.1  627.96   308.2  631.16   388.5  630.69
   404.6  632.53   420.6  637.93   432.7  638.76     501   638.5   537.1  636.11
   553.2  633.38   573.3  637.39   605.4  635.69   609.4  637.08   613.4   640.5
   621.4   652.6   625.5  655.38   645.5   660.6   669.6  664.54     697  665.97
#Mann= 6, -1 ,  0
       0    0.08       0   235.9   0.045       0   292.1    0.05       0
  344.31    0.06       0  444.31    0.05       0  544.31    0.06       0
Bank Sta=235.9,292.1
XS Rating Curve= 0 ,0
Exp/Cntr(USF)=0,0
Exp/Cntr=0.3,0.1

Type RM Length L Ch R = 1 ,5135    ,65.7,65.4,65
XS GIS Cut Line= 2
1597321.01774741 440314.275088911598057.01214977440266.558359484
#Sta/Elev= 30
       0  745.07    11.1  737.22    55.2  716.58    83.3  699.06    99.3   687.1
   131.4   671.2   139.4  663.64   147.4  649.68   155.4  643.87   179.5  636.02
   247.6  627.17   287.7  626.18   301.5  627.27   311.7  632.13   315.8  632.51
   347.8  632.78   403.9  630.41     412  631.96     428  637.42   441.2   638.3
   485.8  638.86   548.2     637   576.3  637.78   600.4   636.3   604.4  637.47
   608.4  641.05   616.4  653.34   620.4  655.11   656.5  658.15   737.5  671.64
#Mann= 5, -1 ,  0
       0    0.08       0   247.6   0.045       0   301.5    0.06       0
     450    0.05       0     550    0.06       0
Bank Sta=247.6,301.5
XS Rating Curve= 0 ,0
Exp/Cntr(USF)=0,0
Exp/Cntr=0.3,0.1

Type RM Length L Ch R = 1 ,5070    ,326.7,328.1,327.9
XS GIS Cut Line= 2
1597310.89601693440382.2352793041598074.36368774440327.288742389
#Sta/Elev= 30
       0  773.31     9.2  764.69    37.3   742.9    81.4   717.1    97.5  700.74
   145.6  663.87   149.6  659.34   157.6  643.76   161.6  640.11   198.3  638.78
   221.8  636.03   233.8   637.6   241.8  628.84   245.9  627.19   269.9  626.92
   281.9  626.12     314  626.97   326.1  631.85   414.3  630.69   438.3  636.28
   474.4  638.81   574.7  636.11   618.8  636.78   622.8  639.38   634.9  655.07
   642.9  659.77     683  665.56   743.1  670.06     760  669.85   765.4  670.29
#Mann= 7, -1 ,  0
       0     0.1       0      70    0.08       0   269.9   0.045       0
     314    0.06       0     460    0.05       0     560    0.06       0
     760     0.1       0
Bank Sta=269.9,314
XS Rating Curve= 0 ,0
Exp/Cntr(USF)=0,0
Exp/Cntr=0.3,0.1

Type RM Length L Ch R = 1 ,4742    ,407.7,414.7,417.3
XS GIS Cut Line= 4
1597320.44986494440598.3829138391597397.70804785440695.795405339
1598166.93082555 440665.563942461598553.22174012440672.282045322
#Sta/Elev= 30
       0  759.86   102.5  729.86   150.8  709.89   202.8  694.43   234.8   666.9
   238.8  664.76   258.8  664.92   266.8  662.78   274.9  656.53   286.9  651.09
   313.1 627.533   318.9  625.32   346.9  625.13   362.9  625.53   369.2 627.464
     415  630.38     467  630.45     487  636.15     511  639.59   679.2  640.07
   731.2  641.91   755.2  649.13   775.2  651.08   791.3   659.4   879.3  680.89
  1014.5  708.88  1055.5  719.55  1110.6  727.86  1235.4  762.85  1280.5  770.53
#Mann= 8, -1 ,  0
       0     0.1       0  204.33    0.05       0  304.33     0.1       0
   313.1   0.045       0   369.2     0.1       0  404.33    0.06       0
  504.33    0.05       0  694.33    0.08       0
Bank Sta=313.1,369.2
XS Rating Curve= 0 ,0
Exp/Cntr(USF)=0,0
Exp/Cntr=0.3,0.1

Type RM Length L Ch R = 1 ,4327    ,66.4,64.8,63.9
XS GIS Cut Line= 2
1597332.09152861441004.3867051561598023.58501991441158.286171208
#Sta/Elev= 30
       0  669.22     4.1  667.93    32.8  668.21    57.4  660.57    90.2  654.93
   106.6  653.66     123  654.44   258.2  642.81   278.7  637.19   299.2  634.59
   315.6  627.85     332  625.86   348.3  623.64   368.9  624.06   383.4625.9244
   392.3   629.3   397.5  629.68   439.2  627.98   463.1  628.98   483.6  627.04
   487.7  628.33   502.9  637.75   508.2  639.42   546.5  640.66   549.9  641.95
   569.6  655.54   583.4  661.09   603.5  662.84   684.4  662.46   708.4  667.96
#Mann= 9, -1 ,  0
       0    0.05       0     150    0.06       0     250    0.05       0
     332   0.045       0   383.4     0.1       0     450    0.06       0
     550    0.07       0     650    0.05       0     690    0.07       0
#XS Ineff= 2 , 0
                          456.58          640.46
Permanent Ineff=
       F       F
Bank Sta=332,383.4
XS Rating Curve= 0 ,0
Exp/Cntr(USF)=0,0
Exp/Cntr=0.3,0.1
